--- 4078_ras.prj (project) ---

Proj Title=4078
Current Plan=p01
Default Exp/Contr=0.3,0.1
English Units
Geom File=g01
Flow File=f01
Plan File=p01
Y Axis Title=Elevation
X Axis Title(PF)=Main Channel Distance
X Axis Title(XS)=Station
BEGIN DESCRIPTION:
RFD model 4078 exported to HEC-RAS
END DESCRIPTION:

--- 4078_ras.p01 (plan) ---

Plan Title=Plan 01
Program Version=4.10
Short Identifier=Plan 01
Geom File=g01
Flow File=f01
Subcritical Flow
Calc Critical at every XS
Secant Critical Depth

--- 4078_ras.f01 (steady flow) ---

Flow Title=Flow 01
Program Version=5.01
Number of Profiles= 6
Profile Names=10yr,25yr,50yr,100yr,100plus,500yr
River Rch & RM=4078,124,31952.86
  103.83  181.94  260.53  340.41     497  1017.3
River Rch & RM=4078,124,30666.08
  147.77  259.93  373.25  488.68  713.47 1393.39
River Rch & RM=4078,124,30568.18
  151.88  267.29  383.95  502.81   734.1  1428.7
River Rch & RM=4078,124,30372.38
  153.93  270.95  389.27  509.85  744.37 1446.23
River Rch & RM=4078,124,30274.47
  156.73  275.98  396.57  519.49  758.45  1470.2
River Rch & RM=4078,124,30176.57
  160.04  281.88  405.16  530.84  775.02 1498.33
River Rch & RM=4078,124,30078.67
  161.05   283.7  407.79  534.32  780.11 1506.95
River Rch & RM=4078,124,29882.87
  162.06  285.51  410.42   537.8  785.18 1515.54
River Rch & RM=4078,124,29687.06
  180.73  318.83  458.78  601.61  878.35 1671.29
River Rch & RM=4078,124,29589.16
  185.63  327.62  471.57  618.52  903.04  1712.4
River Rch & RM=4078,124,29491.26
  248.41  439.26  633.21   831.3  1213.7 2211.14
River Rch & RM=4078,124,29393.36
  249.92  442.02  637.27  836.73 1221.62 2224.08
River Rch & RM=4078,124, 29158.2
  254.45  450.28  649.44  852.97 1245.34 2262.72
River Rch & RM=4078,124,29008.97
   297.5  528.45  764.17 1005.81 1468.49 2618.78
River Rch & RM=4078,124,28859.73
  298.51  530.31  766.92 1009.51 1473.88 2627.43
River Rch & RM=4078,124,28710.49
  299.53  532.18  769.68  1013.2 1479.27 2636.07
River Rch & RM=4078,124,28561.26
  304.78  541.83  783.96 1032.36 1507.24 2680.82
River Rch & RM=4078,124,28412.02
   309.4  550.33  796.53 1049.22 1531.87 2720.16
River Rch & RM=4078,124,28208.72
  314.21  559.18  809.62 1066.78  1557.5 2760.98
River Rch & RM=4078,124,27869.59
  315.81  562.12  813.98 1072.62 1566.03 2774.53
River Rch & RM=4078,124,27666.94
  317.19  564.67  817.76  1077.7 1573.44 2786.37
River Rch & RM=4078,124,27419.64
  320.93  571.56  827.98 1091.45 1593.52  2818.4
River Rch & RM=4078,124,27172.35
  399.23  712.95 1034.82 1366.08 1994.48 3427.74
River Rch & RM=4078,124,26925.06
  402.32  718.79 1043.63  1378.1 2012.02 3455.74
River Rch & RM=4078,124,26677.77
  403.34  720.74 1046.56  1382.1 2017.86 3465.05
River Rch & RM=4078,124,26430.48
  407.11  727.87 1057.32 1396.76 2039.27 3499.11
River Rch & RM=4078,124,26183.18
  411.83  736.75 1070.64 1414.86 2065.69 3540.73
River Rch & RM=4078,124,25798.67
  415.76  744.19 1081.84 1430.12 2087.97 3576.03
River Rch & RM=4078,124,25560.25
     417  746.51 1085.32 1434.82 2094.84 3586.75
River Rch & RM=4078,124, 25258.2
  418.48  749.34 1089.61  1440.7 2103.43 3600.51
River Rch & RM=4078,124,24983.78
  419.01  750.33  1091.1 1442.72 2106.36 3605.09
River Rch & RM=4078,124,24787.62
  505.01  908.47 1325.21 1756.82 2564.95 4293.38
River Rch & RM=4078,124,24458.28
  508.51  915.15 1335.32 1770.64 2585.14  4324.7
River Rch & RM=4078,124, 24323.5
  514.68  926.83 1352.94 1794.67 2620.22 4378.59
River Rch & RM=4078,124,24078.45
  519.96  937.05 1368.55 1816.19 2651.63 4428.01
River Rch & RM=4078,124,23833.39
  521.33  939.69 1372.58 1821.73 2659.73 4440.68
River Rch & RM=4078,124,23588.34
  534.45  964.78 1410.61 1873.84  2735.8 4558.26
River Rch & RM=4078,124,23343.29
   539.9  975.27 1426.61 1895.85 2767.94 4608.29
River Rch & RM=4078,124,23098.23
  542.62  980.51 1434.59 1906.84 2783.98 4633.23
River Rch & RM=4078,124,22853.18
  550.49  995.84 1458.08 1939.32 2831.41 4707.72
River Rch & RM=4078,124,22608.12
  555.41 1005.43  1472.8 1959.69 2861.14 4754.38
River Rch & RM=4078,124,22363.07
  563.42 1021.17 1497.06  1993.4 2910.36 4832.21
River Rch & RM=4078,124,22118.01
  566.15 1026.58 1505.45  2005.1 2927.44 4859.41
River Rch & RM=4078,124,21872.96
  569.44 1033.08 1515.51 2019.12 2947.92 4891.96
River Rch & RM=4078,124,21627.91
  571.62  1037.4 1522.19 2028.45 2961.54 4913.61
River Rch & RM=4078,124,21382.85
  671.63 1225.19 1804.05 2411.16  3520.3  5736.6
River Rch & RM=4078,124,21220.05
  672.55 1227.01 1806.87  2415.1 3526.05 5745.51
River Rch & RM=4078,124, 21099.9
  673.08 1228.05 1808.48 2417.35 3529.33  5750.6
River Rch & RM=4078,124,20644.12
   673.6 1229.09 1810.09  2419.6 3532.61 5755.68
River Rch & RM=4078,124,20397.29
  676.37 1234.56 1818.55 2431.39 3549.83 5782.34
River Rch & RM=4078,124,20150.45
  687.26 1256.09 1851.88 2477.88  3617.7 5887.25
River Rch & RM=4078,124,19903.61
  688.02  1257.6 1854.24 2481.19 3622.53 5894.81
River Rch & RM=4078,124,19656.77
  688.85  1259.3 1856.92 2484.97 3628.06 5903.62
River Rch & RM=4078,124,19409.94
  699.07 1279.64 1888.53 2529.21 3692.65 6003.94
River Rch & RM=4078,124, 19163.1
  699.88 1281.31 1891.17 2532.95 3698.11 6012.68
River Rch & RM=4078,124,18916.26
  730.94 1342.28 1985.22 2663.74 3889.07  6303.5
River Rch & RM=4078,124,18669.43
  826.13 1532.53  2281.9 3080.17 4497.05 7236.07
River Rch & RM=4078,124,18422.59
  925.52 1729.91 2588.76  3509.9 5124.45  8174.5
River Rch & RM=4078,124,18175.75
  929.39 1737.83 2601.29  3527.7 5150.45 8214.32
River Rch & RM=4078,124,17928.92
  932.68 1744.59    2612 3542.95 5172.71 8248.55
River Rch & RM=4078,124,17682.08
  936.26 1751.95 2623.68 3559.61 5197.03 8286.03
River Rch & RM=4078,124,17435.24
  936.88 1753.23 2625.73 3562.54 5201.31 8292.64
River Rch & RM=4078,124,17188.41
  942.52    1765 2644.56 3589.55 5240.75 8354.21
River Rch & RM=4078,124,16941.57
  953.12 1787.16 2680.04 3640.49 5315.12 8470.26
River Rch & RM=4078,124,16694.73
  953.69 1788.37    2682 3643.32 5319.25 8476.81
River Rch & RM=4078,124,16447.89
  964.22  1810.6  2717.8 3694.97 5394.65 8595.46
River Rch & RM=4078,124,16201.06
  970.45 1823.77 2739.03 3725.62 5439.41 8665.91
River Rch & RM=4078,124,15954.22
   971.4 1825.78 2742.28 3730.32 5446.26 8676.72
River Rch & RM=4078,124,15707.38
  972.52 1828.18 2746.16 3735.94 5454.47  8689.7
River Rch & RM=4078,124,15460.55
  999.07  1885.4 2839.39 3871.69 5652.67 9006.33
River Rch & RM=4078,124,14961.82
 1004.05 1896.22 2857.09 3897.57 5690.45    9067
River Rch & RM=4078,124,14606.44
 1005.01  1898.3  2860.5 3902.56 5697.73 9078.69
River Rch & RM=4078,124,14213.73
 1010.29 1909.87 2879.52 3930.45 5738.46 9144.48
River Rch & RM=4078,124,13789.59
 1012.72 1915.16 2888.17  3943.1 5756.93 9174.12
River Rch & RM=4078,124,13440.84
 1014.67 1919.43  2895.2 3953.42 5771.99 9198.45
River Rch & RM=4078,124,13126.58
  1016.6 1923.74 2902.36    3964 5787.45  9223.8
River Rch & RM=4078,124, 12999.4
 1018.72 1928.44 2910.15 3975.51 5804.24 9251.24
River Rch & RM=4078,124,12717.55
 1019.75 1930.77 2914.01 3981.22 5812.58 9264.95
River Rch & RM=4078,124,12630.99
 1020.38 1932.17 2916.36 3984.71 5817.68 9273.38
River Rch & RM=4078,124,12050.42
 1023.02 1938.15 2926.34 3999.54 5839.33 9309.18
River Rch & RM=4078,124,11428.01
 1024.99 1942.58 2933.72 4010.48  5855.3 9335.46
River Rch & RM=4078,124,11178.23
 1025.69 1944.16 2936.36  4014.4 5861.03 9344.92
River Rch & RM=4078,124,10928.45
 1028.67 1950.86 2947.53 4030.97 5885.22 9384.81
River Rch & RM=4078,124,10678.68
 1029.37 1952.44 2950.17 4034.89 5890.94 9394.25
River Rch & RM=4078,124, 10428.9
  1030.2 1954.34 2953.35 4039.64 5897.87 9405.77
River Rch & RM=4078,124,10179.12
 1031.48 1957.27 2958.27 4046.97 5908.58 9423.58
River Rch & RM=4078,124,9929.349
 1066.69 2035.44  3087.8 4238.28 6187.89 9877.93
River Rch & RM=4078,124,9679.573
 1067.29 2036.81 3090.09 4241.69 6192.87 9886.16
River Rch & RM=4078,124,9429.797
 1071.61 2046.57 3106.43 4266.01 6228.38 9944.66
River Rch & RM=4078,124,9180.021
 1073.13    2050 3112.17 4274.55 6240.84 9965.15
River Rch & RM=4078,124,8930.245
 1075.43 2055.18 3120.81 4287.38 6259.58 9995.86
River Rch & RM=4078,124,8680.468
 1179.94 2284.71 3499.52 4845.31 7074.1611297.53
River Rch & RM=4078,124,8430.692
 1182.33 2290.06 3508.44 4858.56  7093.511328.72
River Rch & RM=4078,124,8180.916
 1189.53 2306.24 3535.49 4898.85 7152.3211424.01
River Rch & RM=4078,124, 7931.14
 1190.75 2308.94 3539.97 4905.49 7162.0111439.54
River Rch & RM=4078,124,7681.364
 1197.75 2324.58 3566.04 4944.22 7218.5611530.61
River Rch & RM=4078,124, 7437.15
 1199.27 2327.95 3571.63  4952.5 7230.6511549.95
River Rch & RM=4078,124,7159.664
  1200.4 2330.47 3575.82 4958.71 7239.7211564.44
River Rch & RM=4078,124,6815.037
  1214.1 2360.78  3626.1 5033.16 7348.4111737.84
River Rch & RM=4078,124,6144.671
  1216.9 2366.75  3635.8 5047.28 7369.0311769.53
Boundary for River Rch & Prof#=4078,124,1
Up Type= 0
Dn Type= 2
Boundary for River Rch & Prof#=4078,124,2
Up Type= 0
Dn Type= 2
Boundary for River Rch & Prof#=4078,124,2
Up Type= 0
Dn Type= 2
Boundary for River Rch & Prof#=4078,124,2
Up Type= 0
Dn Type= 2
Boundary for River Rch & Prof#=4078,124,2
Up Type= 0
Dn Type= 2
Boundary for River Rch & Prof#=4078,124,2
Up Type= 0
Dn Type= 2

--- 4078_ras.g01 (geometry) ---

Geom Title=4078
Program Version=4.10

River Reach=4078,124
Reach XY= 30
665827.460793167743571.431197882665463.623225063742682.934198871
665692.912182063741724.643003449665320.082320929741072.733281225
 665492.39134869740613.097864553666435.533709794 738787.57703121
666902.981626511738568.393003419667218.085793138737414.313142315
668268.867043138736547.125642329668702.894820929 736553.20203121
669981.106626481734816.309670091671430.585793167733512.663836762
671782.148293167732687.143003419671645.169126481731959.018003434
672009.231626511731937.143003434671824.335793138731225.163836762
672605.585793138731119.434670091672899.335793167730429.330503419
672887.877459854730774.643003434673078.502459824730795.476336747
674454.023293167730335.580503419675200.898293138729853.288836762
675570.038918167  729166.6568923676986.705584854728993.913836762
677518.838564306728519.396749184677662.935786486727624.431471422
676879.949675381726669.570360303676608.682314277 725513.97140196
675296.833355933725393.528693631674645.791689277724396.349874184

Type RM Length L Ch R = 1 ,31952.86,111.959800,111.959800,111.959800
XS GIS Cut Line= 5
665927.854630015743580.572775296665842.641331471743570.704445885
665828.443405749743570.414107662665826.443702948  743570.4485853
665726.472906496743569.187478623
#Sta/Elev= 26
9899.016745.5589 9901.89744.68589911.957742.92589922.024744.55599932.091 747.919
9942.157749.69829947.459749.36919952.224749.11139962.291747.08649972.358742.8708
9982.425737.21789984.799735.85889992.442731.2008    9999729.6787   10001729.2029
10002.44728.857410012.44731.147710022.45737.748710032.45745.479710042.45749.9839
10052.45 754.13910062.45756.862710072.45758.970510082.45759.906610092.45 759.775
10100.98760.3097
#Mann= 3 , 0 , 0
9899.016    0.04       09899.016    0.04       010100.98    0.04       0
#XS Ineff= 2 , 0
       0                               0
Bank Sta=9899.016,10100.98
Exp/Cntr=0.3,0.1

Type RM Length L Ch R = 1 , 31840.9,97.901700,97.901700,97.901700
XS GIS Cut Line= 4
665962.529220372743470.926275879665919.596658856743464.363940358
665791.585995972743465.647395119665691.721129388743481.934734851
#Sta/Elev= 25
9879.986744.52899887.603742.40849897.719738.09529907.835739.64819917.951737.5967
9923.417734.83519938.015 729.2899948.015727.76049958.016727.23449978.017727.0448
9988.017726.727410018.02725.979810048.02726.234710051.43726.555210058.11727.9538
10068.24731.355510078.37735.1952 10088.5736.501110098.64735.839510108.77735.4431
 10118.9736.187610129.03737.987310139.16740.1181 10149.3742.070910152.62742.9058
#Mann= 3 , 0 , 0
9879.986    0.04       09879.986    0.04       010152.62    0.04       0
#XS Ineff= 2 , 0
       09976.977        10026.59       0
Bank Sta=9879.986,10152.62
Exp/Cntr=0.3,0.1

Type RM Length L Ch R = 1 ,   31743,97.901700,97.901700,97.901700
XS GIS Cut Line= 6
665905.262667263743370.740374481665828.849685924743380.795675622
 665814.03907273743379.932000891665791.107362125743374.350769539
665772.590130165743374.290734983665706.367902327743388.477161938
#Sta/Elev= 27
9899.047713.76769899.313713.79599919.552722.73289929.672725.64859939.791725.0439
9949.903721.86989959.942716.51549969.982711.43249976.156708.11649980.012705.7754
9990.029698.9027    9999 692.50310000.39 691.671   10001691.945710010.65697.9284
10014.63701.493110020.73706.566510030.73711.963210033.14712.778410040.83715.6511
10050.96719.058610061.14723.135910071.44727.052110081.73729.629410086.37730.0891
10092.03730.424610100.92730.8013
#Mann= 3 , 0 , 0
9899.047    0.04       09899.047    0.04       010100.92    0.04       0
#XS Ineff= 2 , 0
       0                               0
Bank Sta=9899.047,10100.92
Exp/Cntr=0.3,0.1

Type RM Length L Ch R = 1 , 31645.1,97.901700,97.901700,97.901700
XS GIS Cut Line= 6
 665873.95041784743256.320057089665810.579702512743276.761815904
665793.707044325743288.056738394665777.339246033743308.615837624
665762.970378726  743319.7881987665697.014050018743343.559550517
#Sta/Elev= 27
9899.138725.77349908.418720.71229918.788715.77599929.157711.16889939.527706.1765
9950.296701.85219961.076 697.0639965.825 694.8369980.634688.63669986.129685.8923
9995.166682.0139    9999681.14019999.924681.1034   10001681.383310007.81685.1125
10012.43689.257410015.39691.676310022.83696.616410028.06699.079410039.36702.7654
10050.32707.295710058.77710.214510061.16710.998210071.62713.005510082.07 715.911
10092.52720.277610100.87722.9633
#Mann= 3 , 0 , 0
9899.138    0.04       09899.138    0.04       010100.87    0.04       0
#XS Ineff= 2 , 0
       0                               0
Bank Sta=9899.138,10100.87
Exp/Cntr=0.3,0.1

Type RM Length L Ch R = 1 , 31547.2,97.901700,97.901700,97.901700
XS GIS Cut Line= 6
665884.020034827743193.187111439665821.527983672743204.045948135
 665785.09492804743206.694779183 665783.09532792 743206.65478718
665729.239933088743209.454200493665683.819870288743216.919366903
#Sta/Elev= 29
9899.042723.93349908.198718.08699909.632 717.1699918.347711.68859928.497707.0325
9938.647702.68179948.797696.67479958.947693.48629962.471692.10529969.016689.2398
9975.628685.65419979.042683.77269989.069675.9303    9999669.41689999.095669.3506
   10001670.056210009.11673.184710019.12679.060510029.13685.781610039.15689.7033
10049.16692.682710054.93693.947810059.22695.096910069.36699.024610079.49702.5578
10089.12704.590210089.63704.712510099.76 709.34510100.96709.7202
#Mann= 3 , 0 , 0
9899.042    0.04       09899.042    0.04       010100.96    0.04       0
#XS Ineff= 2 , 0
       0                               0
Bank Sta=9899.042,10100.96
Exp/Cntr=0.3,0.1

Type RM Length L Ch R = 1 ,31449.29,97.901700,97.901700,97.901700
XS GIS Cut Line= 6
665850.235285386743067.671882772 665796.00683211743093.152669625
665760.623564722743111.958956606665758.763951496743112.695053508
665707.138544366743141.927256343665670.676556905743159.923081163
#Sta/Elev= 27
9899.013713.02069904.797 712.1349915.846710.66869916.244710.55529926.895706.2668
9937.944700.23369939.759698.63169948.993694.6373 9960.07692.74439962.866691.9966
9971.394686.70379984.173674.14859994.044662.6179    9999661.0947   10001661.0447
10005.33661.937810016.82669.308810028.31676.1781 10039.8681.351210046.27683.6316
10051.29685.605210060.33689.630310062.71690.823410067.27692.384810085.02699.0518
10096.17701.448110100.99702.1685
#Mann= 3 , 0 , 0
9899.013    0.04       09899.013    0.04       010100.99    0.04       0
#XS Ineff= 2 , 0
       0                               0
Bank Sta=9899.013,10100.99
Exp/Cntr=0.3,0.1

Type RM Length L Ch R = 1 ,31351.39,97.901700,97.901700,97.901700
XS GIS Cut Line= 6
 665780.13225814742980.989138447665715.492577777743018.616486447
665704.814822323743028.370612319 665692.45889345743046.977943129
665679.928526393743059.839617305665621.442536411743102.269372102
#Sta/Elev= 28
9899.091697.17759905.029695.06019907.063693.6187  9916.6688.89329926.941685.7499
9928.171 685.5939939.742685.47239946.818683.96259951.313682.68579962.884677.3212
9966.696 675.9029974.552672.54749983.349667.94019988.347662.43189996.387654.3646
    9999654.6706   10001655.077810006.09656.673110008.32657.937510021.38667.1482
10028.65 672.69810036.97 678.85110047.67687.9165 10053.1691.397310060.39694.4317
 10070.2697.993110072.48698.635110100.95700.5319
#Mann= 3 , 0 , 0
9899.091    0.04       09899.091    0.04       010100.95    0.04       0
#XS Ineff= 2 , 0
       0                               0
Bank Sta=9899.091,10100.95
Exp/Cntr=0.3,0.1

Type RM Length L Ch R = 1 ,31253.49,97.901700,97.901700,97.901700
XS GIS Cut Line= 6
665732.569671109742885.634767248665703.437272592742906.295832609
665682.595816972742924.952710738665653.259566482742968.151081855
 665642.55264092742980.336518044665587.866238312 743023.24522446
#Sta/Elev= 28
9899.072 686.8029908.352 687.2119915.261687.27879920.612686.32419934.787682.7832
9946.111677.37849947.837676.34629959.533 670.7489962.821669.54489974.743666.7233
 9975.75666.24769986.292657.44989988.435655.39459991.563652.9354    9999649.4494
9999.951 649.116   10001649.595410015.19659.245710024.31664.419810027.71665.8617
10041.01670.512310053.73676.352110055.17677.286910066.44682.914210071.37685.1228
10079.15687.790910087.57688.908510100.93689.1837
#Mann= 3 , 0 , 0
9899.072    0.04       09899.072    0.04       010100.93    0.04       0
#XS Ineff= 2 , 0
       0                               0
Bank Sta=9899.072,10100.93
Exp/Cntr=0.3,0.1

Type RM Length L Ch R = 1 ,31155.59,97.901700,97.901700,97.901700
XS GIS Cut Line= 6
665673.523787929742849.720327594665632.931584627742873.243552967
665588.231946237742895.601561923665585.605440605742897.229460563
665584.100287211742898.546469774665498.353736214742949.974004533
#Sta/Elev= 26
9899.015681.76459909.545682.25699920.424682.23879929.489680.24229931.982679.3523
 9943.54674.48449949.857671.5317 9965.98662.74329977.161657.60989988.342 648.133
 9995.91645.8809    9999645.45849999.804645.4797   10001645.950610011.61650.8898
10013.55651.954310023.27659.149710032.99664.093810034.93664.930910046.59669.1758
10052.43671.535110058.25672.512510069.91673.564410081.58 675.51910093.24678.2057
10100.99679.0986
#Mann= 3 , 0 , 0
9899.015    0.04       09899.015    0.04       010100.99    0.04       0
#XS Ineff= 2 , 0
       0                               0
Bank Sta=9899.015,10100.99
Exp/Cntr=0.3,0.1

Type RM Length L Ch R = 1 ,31057.69,97.901700,97.901700,97.901700
XS GIS Cut Line= 6
665632.799709578 742760.70575537665595.599864055742777.136117765
665570.564308642742791.470644847665558.165824188742801.931579262
665524.892435775742838.432032227665468.637114535 742874.05946542
#Sta/Elev= 29
9899.072657.86149907.599659.74289918.531663.39749929.463668.17879934.452669.9374
9939.739671.3482 9940.43671.48739951.953 671.7919955.565670.49429963.477666.6324
9968.588663.88789974.061661.15999975.868 660.032 9984.81652.59199989.757647.8138
    9999642.2534   10001641.9275 10001.7641.889910005.65644.063510014.62651.2236
 10020.5653.548510029.29655.686910046.36660.281310058.53664.954910070.36668.5688
10081.96669.017310083.09668.578510093.57665.331610100.95662.0973
#Mann= 3 , 0 , 0
9899.072    0.04       09899.072    0.04       010100.95    0.04       0
#XS Ineff= 2 , 0
       0                               0
Bank Sta=9899.072,10100.95
Exp/Cntr=0.3,0.1

Type RM Length L Ch R = 1 ,30959.79,97.901700,97.901700,97.901700
XS GIS Cut Line= 6
665620.665541656742700.945089003665559.618616079742719.109768918
665523.990315104742725.936752203 665522.00972715742726.214729461
665506.852638822742729.861224072665434.039648648742772.319109048
#Sta/Elev= 30
9899.031648.83299904.942645.34159913.249652.87029915.376655.14339925.809663.8246
9936.242667.17069946.676668.66019948.313668.27799957.109 665.7989967.426658.6559
9977.608650.9243 9987.79645.17539994.022639.91489997.972636.4244   10001638.0881
10008.21642.269510016.59644.397210018.73645.061410026.79646.661810030.31647.5469
10041.89648.931910046.64649.067410053.46648.248610065.04636.6521 10066.5636.3481
10076.61639.447210086.35647.270210088.19648.423910099.77 654.21810100.88654.8484
#Mann= 3 , 0 , 0
9899.031    0.04       09899.031    0.04       010100.88    0.04       0
#XS Ineff= 2 , 0
       0                10028.59       0
Bank Sta=9899.031,10100.88
Exp/Cntr=0.3,0.1

Type RM Length L Ch R = 1 ,30861.88,97.901700,97.901700,97.901700
XS GIS Cut Line= 6
665556.627793355742640.995658264665519.366296883742654.081067952
665477.196903326742675.844987111665464.389840093742677.312135366
665427.868182194742680.743858923665363.586260747742692.194191072
#Sta/Elev= 25
9899.162658.25629911.486663.89299922.085665.08389932.684662.39879940.658658.7295
9943.568 657.3219954.822  651.659962.463648.41629966.075645.30179977.328641.7304
9984.267638.9707 9988.32636.96819998.386627.0629   10001627.984610008.43631.0562
10018.47643.514310028.52651.558810035.69655.2393 10038.6656.863610048.76661.3069
10058.91663.629410069.07666.215710079.23666.638210089.39667.589210100.98668.4095
#Mann= 3 , 0 , 0
9899.162   0.055       09899.162   0.055       010100.98   0.055       0
#XS Ineff= 2 , 0
       0                               0
Bank Sta=9899.162,10100.98
Exp/Cntr=0.3,0.1

Type RM Length L Ch R = 1 ,30763.98,97.901700,97.901700,97.901700
XS GIS Cut Line= 6
665576.662726282742597.434156867665540.106427477742598.080662416
665510.307805836 742594.87108156 665488.18386163742589.631293664
665445.958298906742572.479339367665379.750708074742563.112843124
#Sta/Elev= 29
9899.075633.26459900.738631.82469910.739641.00069920.741646.38349930.742649.9151
9935.637651.98819940.773653.7963 9950.83654.52259960.888651.47549965.608648.7168
9971.062645.12279981.339 636.8799988.344630.18769991.845626.6146    9999623.9255
9999.399623.8427   10001624.116710002.94624.679510014.05637.602210024.55645.7548
10025.72646.529710034.04 651.42810045.18657.365410055.35659.706510065.51660.1546
10075.57660.265510085.62660.495810095.68660.910810100.95 661.294
#Mann= 3 , 0 , 0
9899.075   0.055       09899.075   0.055       010100.95   0.055       0
#XS Ineff= 2 , 0
       0                               0
Bank Sta=9899.075,10100.95
Exp/Cntr=0.3,0.1

Type RM Length L Ch R = 1 ,30666.08,97.901800,97.901800,97.901800
XS GIS Cut Line= 6
665589.680543707742494.497678974665517.377641041742493.039096469
665489.723226946742493.946060565665487.733152566742494.145068003
665460.156186683 742494.79770586665387.888722908742490.539891139
#Sta/Elev= 26
9899.013653.54939903.695652.56449913.697652.15689923.699652.25439933.701652.7432
9943.703652.63229953.705649.89669963.707644.56889971.331639.7275 9973.71638.2081
9983.715629.8962 9993.72622.2339    9999620.8314   10001620.305910003.73619.5737
10013.74633.392410023.74642.537310028.58645.595710033.75648.827110043.77652.1648
10053.78652.8415 10063.8652.766810073.82 652.97510083.84653.245810093.85 654.046
10100.98654.5339
#Mann= 3 , 0 , 0
9899.013   0.055       09899.013   0.055       010100.98   0.055       0
#XS Ineff= 2 , 0
       0                               0
Bank Sta=9899.013,10100.98
Exp/Cntr=0.3,0.1

Type RM Length L Ch R = 1 ,30568.18,97.901700,97.901700,97.901700
XS GIS Cut Line= 6
 665596.50831719742394.025084705665530.146062223742390.253826496
665511.221314503742393.634291648 665486.95876188742405.039765701
665470.590312062742409.308260013665398.333809344742409.198914641
#Sta/Elev= 27
 9899.09644.27129900.604643.74479910.643639.41999920.682633.75699930.721629.5256
9940.756632.13169950.757 633.4859960.757632.41049965.611631.78679970.838630.8095
9980.997 629.5499984.835625.71429988.216 622.1689991.636618.8117    9999615.7436
10002.74614.984410011.57621.100610013.69 622.43810024.02629.663910028.58632.4852
10034.18635.6845 10044.2639.215810064.23640.530210074.23642.364710084.24 644.372
10094.25645.804910100.92646.4319
#Mann= 3 , 0 , 0
 9899.09    0.04       0 9899.09    0.04       010100.92    0.04       0
#XS Ineff= 2 , 0
       0                               0
Bank Sta=9899.09,10100.92
Exp/Cntr=0.3,0.1

Type RM Length L Ch R = 1 ,30470.28,97.901700,97.901700,97.901700
XS GIS Cut Line= 6
665616.237243743742336.614317276665561.911440081742325.760453113
665519.373118145742312.475620453665517.486742068742311.811101606
 665475.33102419742297.487188594665421.208289313742285.495279162
#Sta/Elev= 27
9899.036648.60819907.276646.73289910.495646.13949920.693643.14379930.891639.0764
9941.088637.38369951.286 634.5519956.986630.49759961.676627.37269972.152620.8127
9982.629614.99429993.105606.5115    9999605.2036   10001604.964310003.63604.8144
10014.19612.961310022.17615.575610024.75616.197910035.31615.654410045.86608.4811
 10056.1606.105310057.02606.015110066.35607.863310076.59611.981610086.83613.2145
10097.07615.546910100.96617.5818
#Mann= 3 , 0 , 0
9899.036   0.055       09899.036   0.055       010100.96   0.055       0
#XS Ineff= 2 , 0
       0                10025.48       0
Bank Sta=9899.036,10100.96
Exp/Cntr=0.3,0.1

Type RM Length L Ch R = 1 ,30372.38,97.901700,97.901700,97.901700
XS GIS Cut Line= 5
665631.199958089742224.543357323665531.599749828742215.632419221
665529.604980236742215.487870699665520.807593989742214.860214466
665429.750107323742210.251511926
#Sta/Elev= 26
9899.002639.71779905.227 637.6469915.267632.26349925.307630.59949935.347630.7601
9945.386632.58529955.426633.45669965.466629.44029975.506 620.9949985.546612.2956
9995.586601.8078    9999602.0318   10001602.202810005.62602.681210007.86604.6399
10009.82606.346310015.63611.371510025.65613.836710035.66615.603910045.67618.1209
10055.69621.2292 10065.7624.804210075.71627.733910085.72630.077610095.74632.8091
10100.99634.1182
#Mann= 3 , 0 , 0
9899.002    0.04       09899.002    0.04       010100.99    0.04       0
#XS Ineff= 2 , 0
       0                               0
Bank Sta=9899.002,10100.99
Exp/Cntr=0.3,0.1

Type RM Length L Ch R = 1 ,30274.47,97.901700,97.901700,97.901700
XS GIS Cut Line= 6
665627.376238008742101.208978441665596.385273799742100.926250931
665566.653989067 742104.99388479665546.893455103742111.342267075
665492.097995131742135.661539879665433.002143693742146.109786801
#Sta/Elev= 28
 9899.08633.87299911.457632.23319921.457630.59499931.471629.16459941.564628.7054
9951.657 627.3489960.101624.68389961.818623.83029972.321617.66779980.836612.3782
9982.921610.9905 9989.57603.45369993.933598.8631    9999598.4601   10001598.5056
10004.91598.941310016.12603.858210021.79606.622910027.07608.938110037.76 611.325
10038.98611.767910048.15615.595110058.43620.4641 10068.7625.471710078.78630.0853
10088.86633.701410098.94635.458410100.96635.1935
#Mann= 3 , 0 , 0
 9899.08   0.055       0 9899.08   0.055       010100.96   0.055       0
#XS Ineff= 2 , 0
       0                               0
Bank Sta=9899.08,10100.96
Exp/Cntr=0.3,0.1

Type RM Length L Ch R = 1 ,30176.57,97.901700,97.901700,97.901700
XS GIS Cut Line= 6
665610.128849243742058.245554608665551.992640943742045.800810622
665513.901576129742032.016737291665512.019186788742031.341007784
665471.328592927742016.538806846665416.540410624742002.041211532
#Sta/Elev= 23
9899.038632.8047 9914.51 630.8159924.736627.59379934.963623.3553 9945.19618.6517
9955.416613.77629960.845610.79369965.928 607.6999976.563 602.9739987.197600.9558
9997.832596.2655    9999 596.484   10001597.013110008.47600.714710019.11610.9152
10029.75615.735810040.39620.671110050.85625.715110061.19629.418910071.53631.3886
10081.88632.880610092.22633.098610100.97633.6838
#Mann= 3 , 0 , 0
9899.038   0.055       09899.038   0.055       010100.97   0.055       0
#XS Ineff= 2 , 0
       0                               0
Bank Sta=9899.038,10100.97
Exp/Cntr=0.3,0.1

Type RM Length L Ch R = 1 ,30078.67,97.901700,97.901700,97.901700
XS GIS Cut Line= 5
665646.826579392741991.105161442665570.964469767741951.050325906
665557.915546124741945.460348493665556.028132963741944.798780993
 665465.17543762741903.112618849
#Sta/Elev= 25
9899.017607.78989901.082606.58899912.391612.55399923.699613.5252 9933.51 612.914
9935.007612.92769946.316610.05779954.928606.72179968.932600.80079976.345598.8753
9980.241597.60449984.804595.01999991.293592.060810000.39591.587310002.13591.4236
10013.13601.239910024.14606.032510035.14608.111110046.14611.796110048.48 612.611
10057.14615.985410068.15621.171110079.15624.609110090.15627.402810100.96628.6847
#Mann= 3 , 0 , 0
9899.017   0.055       09899.017   0.055       010100.96   0.055       0
#XS Ineff= 2 , 0
       0                               0
Bank Sta=9899.017,10100.96
Exp/Cntr=0.3,0.1

Type RM Length L Ch R = 1 ,29980.77,97.901700,97.901700,97.901700
XS GIS Cut Line= 6
665700.062712842741927.842477189665656.865708434 741899.95004973
665618.796422592741869.826400612665581.998034356741841.296857536
665558.875641353741826.961221656665533.541073366741814.593512414
#Sta/Elev= 29
9899.035618.21459905.061616.84449916.964615.0813 9922.71613.59059928.868612.1688
9940.771609.12389952.833603.18499958.431600.94399965.585599.73989974.547598.4034
9978.337597.29359991.089589.6421    9999588.0128   10001588.057510003.77588.4307
10006.93590.046810016.44596.036310023.23599.0069 10029.1600.429610039.53603.4807
10041.76604.214610045.56605.6917 10053.8609.147710057.51610.988210065.56615.6762
10077.08623.203310088.21624.751710099.34 625.23710100.96625.1828
#Mann= 3 , 0 , 0
9899.035    0.04       09899.035    0.04       010100.96    0.04       0
#XS Ineff= 2 , 0
       0                               0
Bank Sta=9899.035,10100.96
Exp/Cntr=0.3,0.1

Type RM Length L Ch R = 1 ,29882.87,97.901700,97.901700,97.901700
XS GIS Cut Line= 6
665759.972015838741827.782714517665706.815497538741805.771143738
665667.416186611741785.225966494665637.297489602741770.659649176
665612.511934853741763.428535086665572.328066647 741757.30273041
#Sta/Elev= 28
9899.029621.16559904.411620.31529906.303619.89699915.234618.33869926.058616.1474
9932.441615.20399936.881613.96959947.705610.12949958.608604.65719969.873602.9691
9979.962598.25389981.137597.59099992.402589.2135    9999585.729310001.52584.8472
10003.68584.691310014.79593.112710024.49597.2726 10025.9597.577110036.85601.0541
10047.27606.510410054.66610.867310057.68612.431810060.27613.033210067.87615.1914
10077.99618.6015 10088.1619.694610100.92 619.854
#Mann= 3 , 0 , 0
9899.029    0.04       09899.029    0.04       010100.92    0.04       0
#XS Ineff= 2 , 0
       0                               0
Bank Sta=9899.029,10100.92
Exp/Cntr=0.3,0.1

Type RM Length L Ch R = 1 ,29784.97,97.901700,97.901700,97.901700
XS GIS Cut Line= 6
665767.749323616741662.321433175665731.475258258741669.529554076
665706.383955669741678.858798483665656.205606376741713.365883304
665636.801044249741723.008597195 665582.74485295741734.471402375
#Sta/Elev= 30
9899.091617.76449901.894618.2453 9912.09617.95239922.285616.30279932.481615.6691
9936.074615.09889942.983614.16189953.652610.28959964.441607.76979975.148598.6993
9975.982597.78899984.936590.59929987.745588.46369993.414585.735910000.36583.1168
   10001583.106510009.88585.402410012.88586.808710023.86589.8692 10025.2 590.199
10036.37592.3613 10047.4595.453310052.83597.181210057.79599.003510068.19603.3668
10072.71605.570210078.42608.127310088.52611.216810098.63614.6403 10100.9615.0122
#Mann= 3 , 0 , 0
9899.091   0.055       09899.091   0.055       0 10100.9   0.055       0
#XS Ineff= 2 , 0
       0                               0
Bank Sta=9899.091,10100.9
Exp/Cntr=0.3,0.1

Type RM Length L Ch R = 1 ,29687.06,97.901700,97.901700,97.901700
XS GIS Cut Line= 6
665727.452474298741614.884595836665653.016076729 741622.45093103
665627.940074813741620.959712463665625.971820778741620.604781408
665589.572136606741617.953837475665526.225383372741621.257915174
#Sta/Elev= 27
 9899.06604.35779900.201604.29349901.525604.17369911.576603.41549921.628602.3692
9931.679602.01919941.731599.57989951.782595.48869961.834588.60839971.886586.6633
 9973.88586.4444 9981.91585.41629991.928584.8635    9999583.1147   10001582.5754
10001.97  582.33   10012584.894610022.03597.837910032.05603.0966 10037.5 604.052
10042.07604.970310052.09605.9843 10062.1606.882310072.12608.335910082.13610.2007
10092.14611.901810100.93 613.696
#Mann= 3 , 0 , 0
 9899.06  0.0497       0 9899.06  0.0497       010100.93  0.0497       0
#XS Ineff= 2 , 0
       0                               0
Bank Sta=9899.06,10100.93
Exp/Cntr=0.3,0.1

Type RM Length L Ch R = 1 ,29589.16,97.901700,97.901700,97.901700
XS GIS Cut Line= 6
 665756.38465723741540.142188089665693.096032915741536.024842075
665637.332207571741522.601298931665611.963667879741518.747825457
665584.779466237 741517.78089512665556.686639737741520.094630822
#Sta/Elev= 18
9899.025607.82469930.426 606.8789940.459606.86399950.519 606.0949960.579601.5109
9970.741595.27339980.927589.622810001.63580.051310010.48583.211710011.97583.8882
 10019.9586.927710022.25587.747410032.37588.989710042.48591.357610052.52592.6392
10072.76593.549710082.57594.285410100.94596.1529
#Mann= 3 , 0 , 0
9899.025  0.0495       09899.025  0.0495       010100.94  0.0495       0
#XS Ineff= 2 , 0
       0                               0
Bank Sta=9899.025,10100.94
Exp/Cntr=0.3,0.1

Type RM Length L Ch R = 1 ,29491.26,97.901700,97.901700,97.901700
XS GIS Cut Line= 6
665740.671555405741409.888540848665651.835137149741430.423839249
665643.365533007741432.873468064665612.370790324741442.295474055
665585.432938488741452.558198633665549.254472882 741471.29680776
#Sta/Elev= 25
9899.004606.29559904.825605.39339915.089602.3644  9921.7600.06169925.353598.6373
9935.616593.3966 9945.88589.51619956.144586.70719966.408 584.1189976.671 582.268
9986.935580.79699990.183579.96929997.299578.3291   10001578.970710006.06580.1077
10007.77580.585110018.21584.228110028.65 585.01510049.99585.913810060.71587.4309
10065.53588.012710083.24589.219910087.28589.7749 10094.5591.106310100.97592.6006
#Mann= 3 , 0 , 0
9899.004   0.055       09899.004   0.055       010100.97   0.055       0
#XS Ineff= 2 , 0
       0                               0
Bank Sta=9899.004,10100.97
Exp/Cntr=0.3,0.1

Type RM Length L Ch R = 1 ,29393.36,85.917700,85.917700,85.917700
XS GIS Cut Line= 6
665716.208023876741239.369009018665645.895523846741279.733592331
665567.722436935741428.769360244665548.164352387  741443.4379237
665516.714359462741471.039068475665472.503363013 741500.72244589
#Sta/Elev= 30
9841.855610.00279843.248609.5849 9877.84608.70119889.371608.68539900.902609.1042
9913.423608.8511 9922.93 608.257 9940.17608.71439946.387608.56139951.462 607.617
9962.754 600.0879974.046585.05989985.338577.11649989.443576.5501 9996.63576.7816
10007.92578.9646 10041.8581.083710053.09581.317510064.38582.707510075.56583.4634
10086.97584.635910094.63585.674710119.88589.9384 10133.2594.023210146.49597.5634
10157.52598.100710171.63599.266710183.67603.599710195.72608.431610210.77610.8198
#Mann= 3 , 0 , 0
9841.855    0.04       09841.855    0.04       010210.77    0.04       0
#XS Ineff= 2 , 0
       0                               0
Bank Sta=9841.855,10210.77
Exp/Cntr=0.3,0.1

Type RM Length L Ch R = 3 , 29336.8,,,
BEGIN DESCRIPTION:
END DESCRIPTION:
Bridge Culvert--1,0,-1,-1, 0
Deck Dist Width WeirC Skew NumUp NumDn MinLoCord MaxHiCord MaxSubmerge Is_Ogee
32.493850,20.930000,2.6,0, 34, 34, , , 0.95, 0, 0,0,,
 9905.73 9913.48 9915.34 9928.04 9929.10 9942.60 9942.86 9955.36 9956.30 9960.47
 9965.15 9966.62 9973.07 9973.07 9975.6910026.3110026.3110029.9710033.1310039.48
10049.3210050.0310058.0410062.9310073.8710075.8310088.7310089.6910101.6310105.52
10114.5310121.3510127.4410132.35
  598.35  597.44  597.23  595.82  595.70  594.07  594.04  592.64  592.56  592.19
  591.71  591.57  590.89  590.89  590.61  588.72  588.72  588.59  588.64  588.73
  589.21  589.25  589.76  590.05  591.27  591.54  593.18  593.30  594.87  595.54
  596.79  597.84  599.07  600.46
 -401.65 -402.56 -402.77 -404.18 -404.30 -405.93 -405.96 -407.36 -407.44 -407.81
 -408.29 -408.43 -409.11  588.39  588.11  586.22 -411.28 -411.41 -411.36 -411.27
 -410.79 -410.75 -410.24 -409.95 -408.73 -408.46 -406.82 -406.70 -405.13 -404.46
 -403.21 -402.16 -400.93 -399.54
 9905.73 9913.48 9915.34 9928.04 9929.10 9942.60 9942.86 9955.36 9956.30 9960.47
 9965.15 9966.62 9973.38 9973.38 9975.6910026.6210026.6210029.9710033.1310039.48
10049.3210050.0310058.0410062.9310073.8710075.8310088.7310089.6910101.6310105.52
10114.5310121.3510127.4410132.35
  598.35  597.44  597.23  595.82  595.70  594.07  594.04  592.64  592.56  592.19
  591.71  591.57  590.85  590.85  590.61  588.71  588.71  588.59  588.64  588.73
  589.21  589.25  589.76  590.05  591.27  591.54  593.18  593.30  594.87  595.54
  596.79  597.84  599.07  600.46
 -401.65 -402.56 -402.77 -404.18 -404.30 -405.93 -405.96 -407.36 -407.44 -407.81
 -408.29 -408.43 -409.15  588.35  588.11  586.21 -411.29 -411.41 -411.36 -411.27
 -410.79 -410.75 -410.24 -409.95 -408.73 -408.46 -406.82 -406.70 -405.13 -404.46
 -403.21 -402.16 -400.93 -399.54
BR Coef=-1 , 0 , 0 ,, 0 ,,,0.8,0,1,0,
WSPro=,,,, 1 ,,,, 0 ,,,, 0 ,,,,-1 ,-1 ,-1 , 0 , 0 , 0 , 0 , 0
BC Design=,, 0 ,, 0 ,,,,,,

Type RM Length L Ch R = 1 ,29307.44,149.236600,149.236600,149.236600
XS GIS Cut Line= 6
665638.083023876741212.025259003665589.905940562741239.369009018
665540.426773846741294.056509018665510.478857219741403.431509018
665419.333023876741455.514842346 665417.62957418 741455.46571283
#Sta/Elev= 30
9812.493606.16169827.536605.39499838.778605.22329850.533604.08689859.037603.8102
9875.482601.74969890.106598.91199902.453595.87459905.011595.54959915.939593.0551
9919.916592.45989929.424 589.9099934.821587.90599942.616586.47569962.187586.4495
 9973.72586.96129984.088576.89539994.456570.765610000.05569.994610004.82569.8363
10015.19575.907810025.56 586.12610035.93590.0402 10058.2591.852610084.38 596.226
 10095.9597.714910118.67600.001610130.45602.122110153.49607.551510161.72608.6671
#Mann= 3 , 0 , 0
9812.493    0.04       09812.493    0.04       010161.72    0.04       0
#XS Ineff= 2 , 0
       0                               0
Bank Sta=9812.493,10161.72
Exp/Cntr=0.3,0.1

Type RM Length L Ch R = 1 , 29158.2,149.236600,149.236600,149.236600
XS GIS Cut Line= 6
665650.946675949741100.393777145665552.491986075 741149.62853008
665499.875269681 741192.52801328 665414.61413308741279.064667567
665329.810970033741338.209953823665243.677848996741385.653533346
#Sta/Elev= 30
9749.074603.44549776.854602.97589821.438603.77379833.136 602.9149850.544600.4002
9893.951599.17899916.001596.47169948.527589.74859959.043 586.7169973.005579.6994
9986.113565.22159992.895562.69559999.212563.0469 10008.4567.819610015.19572.8823
10027.35585.586110035.55591.967710042.85594.870710049.15596.441110059.25598.2847
10085.74600.7988 10098.1602.922410122.34602.517310134.34604.326710158.14604.6001
10169.75606.986610204.56609.517110215.78609.467910238.23610.799410250.94610.5875
#Mann= 3 , 0 , 0
9749.074    0.04       09749.074    0.04       010250.94    0.04       0
#XS Ineff= 2 , 0
       0                               0
Bank Sta=9749.074,10250.94
Exp/Cntr=0.3,0.1

Type RM Length L Ch R = 1 ,29008.97,149.236600,149.236600,149.236600
XS GIS Cut Line= 6
665597.618415031741067.334591544665535.102950304741079.943419693
665478.260726654 741095.78399076665382.162767546 741136.21965385
665258.601306673741181.784342346665121.012292559741220.825814485
#Sta/Elev= 30
 9749.06600.83499787.831601.07829812.941599.16999823.322593.72449833.703591.7937
9864.847590.92449886.036593.25279907.443593.71939929.234 592.5519962.082588.8547
9973.032583.45879983.683563.96659994.216 554.852 10004.7556.9325 10015.2564.1261
10025.92573.821110036.65581.760410047.38588.029310058.11591.859610079.56592.0582
10111.66585.359410122.16585.645610143.15588.427910153.65588.860110184.91593.1138
10215.88593.3094 10226.2590.109710236.52574.929310246.85571.844210250.96573.6155
#Mann= 3 , 0 , 0
 9749.06    0.04       0 9749.06    0.04       010250.96    0.04       0
#XS Ineff= 2 , 0
       0                               0
Bank Sta=9749.06,10250.96
Exp/Cntr=0.3,0.1

Type RM Length L Ch R = 1 ,28859.73,149.236600,149.236600,149.236600
XS GIS Cut Line= 6
665591.302649144741048.921333487665494.776552909 741051.28390792
665420.668723068741042.804364401665380.466423696741030.817380799
665255.720187174740978.564768426665105.630185397740949.054720752
#Sta/Elev= 30
9749.138600.41849775.473600.38879785.485 598.8399805.497594.30289815.497592.5741
9845.497591.62929855.522589.82079875.572585.34539885.615583.88059926.298578.6086
9947.168576.86389957.603576.46799968.421574.45849979.557561.93129990.692552.0155
 9998.29548.871110001.97 548.70710013.05558.424810024.13569.462210034.97578.1639
10045.71581.789210056.44584.208910077.57588.024810108.87591.848410129.42595.1588
 10139.7596.427510160.26598.265910170.54598.676310211.05601.739110250.92604.0859
#Mann= 3 , 0 , 0
9749.138    0.12       09749.138    0.12       010250.92    0.12       0
#XS Ineff= 2 , 0
       0                               0
Bank Sta=9749.138,10250.92
Exp/Cntr=0.3,0.1

Type RM Length L Ch R = 1 ,28710.49,149.236600,149.236600,149.236600
XS GIS Cut Line= 6
665657.674020612740987.533614307665539.043574693740955.992682553
665483.416417302740929.113061021665354.344635019 740851.81657452
665283.149320134 740823.40484497 665197.14744561740797.628342497
#Sta/Elev= 30
9749.117600.62859762.062600.30919772.276599.1748 9782.49599.02499802.917597.3459
9813.174595.42689834.196594.53639855.263592.96469872.071588.43289897.337582.8481
9909.881579.61929932.093572.35079943.673570.15679955.342565.96229967.011562.9044
9980.211557.71799997.749547.988510003.19 546.45710027.09560.117910038.42567.6099
10049.75571.300410077.69573.925310105.57578.216610127.17582.558110148.51584.8082
10169.66587.864810190.42589.030610221.85591.988510242.73592.637410250.93593.8054
#Mann= 3 , 0 , 0
9749.117    0.12       09749.117    0.12       010250.93    0.12       0
#XS Ineff= 2 , 0
       0                               0
Bank Sta=9749.117,10250.93
Exp/Cntr=0.3,0.1

Type RM Length L Ch R = 1 ,28561.26,149.236600,149.236600,149.236600
XS GIS Cut Line= 6
665700.194481437740838.755361155665591.559065509 740781.51116875
665539.770920394740762.038399998665499.147109316 740754.59778575
665383.177563228740745.919423974665221.419536818740708.674214492
#Sta/Elev= 30
9749.087588.84449754.958588.10189766.262582.59889777.565579.03089788.869576.9518
9811.475577.35169842.947584.00719856.689 583.8199871.882580.84399889.837576.1799
 9911.27568.7027 9921.77564.11529942.278551.52689952.444557.0274 9962.61557.4382
9972.714556.17999982.727552.83239992.741548.194610002.75545.856210012.76548.5042
10022.77550.411210032.77 553.44510042.81558.074210062.96566.285210073.03572.0533
 10083.1575.613610093.28 577.86510103.49579.159910154.54582.768110250.96586.6353
#Mann= 3 , 0 , 0
9749.087    0.12       09749.087    0.12       010250.96    0.12       0
#XS Ineff= 2 , 0
       0                               0
Bank Sta=9749.087,10250.96
Exp/Cntr=0.3,0.1

Type RM Length L Ch R = 1 ,28412.02,94.042300,94.042300,94.042300
XS GIS Cut Line= 2
665606.657826781740687.173925757665429.791507334740562.390939638
#Sta/Elev= 24
9865.126 576.9119868.897576.17149879.393573.61179886.243571.38099891.631569.3755
9920.936559.71539928.346557.69449938.283554.75379940.585554.22929952.823 551.971
9955.629551.52779965.061550.1872  9977.3548.86289990.322545.381610001.78543.9166
10007.67548.999310014.01556.851410025.02563.287810026.25563.541710038.49563.6605
10042.36563.794110050.73563.823710075.21565.437810081.58565.9211
#Mann= 3 , 0 , 0
9865.126    0.12       09865.126    0.12       010081.58    0.12       0
#XS Ineff= 2 , 0
       0                10056.56       0
Bank Sta=9865.126,10081.58
Exp/Cntr=0.3,0.1

Type RM Length L Ch R = 1 ,28317.98,109.256100,109.256100,109.256100
XS GIS Cut Line= 3
665655.485951751 740666.55760631 665543.72379896740536.349272981
665425.451229542740462.564550743
#Sta/Elev= 30
9886.356581.36859914.766577.9122 9917.81577.26659927.945574.36699933.163571.5935
9941.123567.82399948.517 564.726 9963.87556.7237 9967.48555.21669979.224 551.317
9980.659550.65999993.837543.09379994.578542.931910007.02543.684510009.93545.0425
10020.19551.009510040.64558.049410046.55559.197910055.99559.151410068.23558.6695
10079.39559.042110098.29553.747410103.59553.611310117.18555.726810127.17558.6202
10138.95562.883610150.74567.883810154.97569.175310162.53570.289510197.35573.7933
#Mann= 3 , 0 , 0
9886.356    0.06       09886.356    0.06       010197.35    0.06       0
#XS Ineff= 2 , 0
       0                10052.83       0
Bank Sta=9886.356,10197.35
Exp/Cntr=0.3,0.1

Type RM Length L Ch R = 1 ,28208.72,339.131500,339.131500,339.131500
XS GIS Cut Line= 5
665730.875324816740543.771565318 665634.10799706740492.107653052
665609.506134033 740508.50889504665567.682966977740505.228646636
 665433.19278267740451.924610183
#Sta/Elev= 30
9914.819581.14489921.479580.41569944.151575.66099954.675571.36759966.823565.0412
9975.908558.8462 9997.14542.821610000.83540.747210012.17545.264710018.37548.9256
 10023.5550.671210035.46550.264610047.48550.537210054.08551.1883 10058.6551.8729
10078.66 553.70510088.69555.208510098.92556.321210109.68556.446710120.43552.9762
10123.79550.994510131.19548.208810141.95551.6316 10152.7555.425410163.46558.7795
10184.97566.456510195.73569.580510206.49571.690110217.24571.8711 10240.7574.6383
#Mann= 3 , 0 , 0
9914.819  0.0405       09914.819  0.0405       0 10240.7  0.0405       0
#XS Ineff= 2 , 0
       0                10022.12       0
Bank Sta=9914.819,10240.7
Exp/Cntr=0.3,0.1

Type RM Length L Ch R = 1 ,27869.59,202.655400,202.655400,202.655400
XS GIS Cut Line= 5
665776.798802316740421.582312509665731.695386857740374.018710732
  665689.0521577740364.177965581665650.509239048740377.298959136
  665533.2403588740329.735357374
#Sta/Elev= 30
9813.339576.4427 9822.41575.78959836.191575.24619849.972572.74329863.754569.5488
9878.887566.85399885.759 566.5279896.021564.09199906.284559.62359916.547558.1237
9918.995558.14769922.651557.48899925.202 557.6319937.495556.73959948.059559.5984
9958.622561.78169963.366561.57739969.311560.50369980.103550.66049990.894539.4242
9996.089536.059710001.69533.319610012.48538.012610023.27548.906310034.06561.3441
10044.85570.4455 10049.3570.745810055.64570.352110066.43570.496610089.91572.5093
#Mann= 3 , 0 , 0
9813.339    0.12       09813.339    0.12       010089.91    0.12       0
#XS Ineff= 2 , 0
       0                               0
Bank Sta=9813.339,10089.91
Exp/Cntr=0.3,0.1

Type RM Length L Ch R = 1 ,27666.94,247.292100,247.292100,247.292100
XS GIS Cut Line= 2
665892.427558303740347.776723579665642.308618009740214.926663488
#Sta/Elev= 30
9884.625580.12849893.035 577.8989911.863572.43659927.004568.96929938.328562.7609
9954.499555.28339960.974552.71569975.817 541.917 9983.62534.90589994.943526.2347
9997.135525.674510006.27525.115910017.59 527.27510028.91532.313710040.24536.9788
10051.56538.944110061.09538.849910062.88539.0469 10074.2541.254210082.41544.3019
10085.53545.142410096.85545.302210103.73548.201110108.17551.2213 10119.5558.5462
10125.04561.646910142.14568.286210146.36570.450110153.47573.440510167.84573.3641
#Mann= 3 , 0 , 0
9884.625    0.04       09884.625    0.04       010167.84    0.04       0
#XS Ineff= 2 , 0
       0                               0
Bank Sta=9884.625,10167.84
Exp/Cntr=0.3,0.1

Type RM Length L Ch R = 1 ,27419.64,247.292000,247.292000,247.292000
XS GIS Cut Line= 6
666068.926336825740197.537601154665982.255200853740161.668020993
665920.422471654740127.795534618665891.438665935740105.533429168
665776.168730936740000.775790749665654.144869317739922.296494064
#Sta/Elev= 30
9749.073572.02079764.145569.79559796.613566.32889818.258562.54539839.903557.3597
9873.312546.41049899.406539.84379918.019536.27949934.436532.37579965.413529.7201
9972.464526.39779980.068519.36489986.144516.23539999.775514.109810009.44517.3663
 10013.5519.787810027.32 532.61710038.43537.016810052.92538.674410054.94539.3783
10068.26548.417410081.28552.8048 10094.3552.771110099.21554.110810107.22557.0914
10131.54569.8907 10143.7574.755810179.73575.583610214.84577.818810250.95576.9301
#Mann= 3 , 0 , 0
9749.073    0.12       09749.073    0.12       010250.95    0.12       0
#XS Ineff= 2 , 0
       0                               0
Bank Sta=9749.073,10250.95
Exp/Cntr=0.3,0.1

Type RM Length L Ch R = 1 ,27172.35,247.292100,247.292100,247.292100
XS GIS Cut Line= 6
666183.756831819739892.019619963666041.754459813739864.261342067
665890.329058539739868.190554825665839.590913581739863.806092888
665770.027209762739845.850611983665693.193690223739815.807590599
#Sta/Elev= 30
 9749.09598.90879778.645598.90719788.923596.55099840.138579.86699860.342574.0071
9870.444 570.3149890.648564.99039900.685560.62719920.695550.00969960.736533.2086
9970.759527.17199980.782518.78969990.806511.489310000.83508.967810010.85 511.755
10020.86520.938110030.87532.749310040.88541.7674 10050.9544.334810060.91545.9538
10091.07554.447210101.22556.084410111.44558.878810121.66563.433110131.96569.7768
10142.38571.089710152.81573.329910170.76575.059810216.78584.968710250.93590.6285
#Mann= 3 , 0 , 0
 9749.09    0.12       0 9749.09    0.12       010250.93    0.12       0
#XS Ineff= 2 , 0
       0                               0
Bank Sta=9749.09,10250.93
Exp/Cntr=0.3,0.1

Type RM Length L Ch R = 1 ,26925.06,247.292100,247.292100,247.292100
XS GIS Cut Line= 6
666232.740274916739743.390679531666100.496804025739684.224554767
666006.611832738739636.959343631666004.827334179739636.056257315
665903.943234329739584.822725956665779.781091057739527.293082793
#Sta/Elev= 30
9749.013  567.629790.358562.07799812.269558.17429834.179554.82959843.017552.5597
9888.955543.65329900.043540.28449944.826530.65249956.022527.17979967.217520.1634
9978.413515.94719989.609506.889810000.81 503.36810003.33 504.06110012.02508.7267
10023.24519.114310025.42520.461710034.45523.682910056.88536.6084 10068.1544.3739
10079.32550.968810112.96551.8971   10124554.859310135.03569.563210146.05577.5883
10168.09578.860110185.09579.1127 10223.2581.911810234.22590.526710250.99598.2815
#Mann= 3 , 0 , 0
9749.013    0.12       09749.013    0.12       010250.99    0.12       0
#XS Ineff= 2 , 0
       0                               0
Bank Sta=9749.013,10250.99
Exp/Cntr=0.3,0.1
